--- ClrFrk1.prj (project) ---

Proj Title=ClrFrk1
Current Plan=p01
Default Exp/Contr=0,0
English Units
Geom File=g01
Flow File=f01
Plan File=p01
BEGIN DESCRIPTION:
END DESCRIPTION:
DSS Export Rating Curves= 0
DSS Export Rating Curve Sorted= 0
DSS Export Volume Flow Curves= 0
DXF OffsetX= 0
DXF OffsetY= 0
DXF ScaleX= 0
DXF ScaleY= 0

--- ClrFrk1.p01 (plan) ---

Plan Title=Floodplain
Program Version=4.00
Geom File=g01
Flow File=f01
K Sum by GR=0
Std Step Tol=0.01
Critical Tol=0.01
Num of Std Step Trials=20
Max Error Tol=0.3
Flow Tol Ratio=0.001
Split Flow NTrial=30
Split Flow Tol=0.02
Split Flow Ratio=0.02
Log Output Level=0
Friction Slope Method=1
Unsteady Friction Slope Method=2
Unsteady Bridges Friction Slope Method=1
Global Log Level=0
CheckData=False
Run HTab=0
Run UNet=0
Run PostProcess=0
UNET Theta=0
UNET Theta Warmup=0
UNET ZTol=0
UNET ZSATol=0
UNET MxIter=0
UNET MaxInSteps=0
UNET DtIC=0
UNET DtMin=0
UNET MaxCRTS=0
UNET WFStab=0
UNET SFStab=0
UNET WFX=0
UNET SFX=0
UNET DSS MLevel=0
UNET DZMax Abort=0
UNET Convert EG Bridges=0
UNET Use Existing IB Tables=0
UNET Froude Limit=0
UNET Froude Power=0
Write IC File=0
Echo Input=False
Echo Output=False
Write Detailed=0

--- ClrFrk1.f01 (steady flow) ---

Flow Title=NFF Regression Equation
Program Version=4.00
Number of Profiles=1
Profile Names=P100yr
River Rch & RM=ClrFrk1,Main      ,51213.8
6495.690
River Rch & RM=ClrFrk1,Main      ,38611.5
6971.407
River Rch & RM=ClrFrk1,Main      ,38038.5
8086.133
River Rch & RM=ClrFrk1,Main      ,32613.8
8230.639
River Rch & RM=ClrFrk1,Main      ,213.8
9141.487
Boundary for River Rch & Prof#=ClrFrk1,Main      ,1
Up Type=0
Dn Type=3
Dn Slope=0.005907

--- ClrFrk1.g01 (geometry) ---

Geom Title=USGS 3m DEM
Program Version=4.10

River Reach=ClrFrk1         ,Main
Reach XY= 30
     1851267.695      344328.957     1849788.545      344028.665
     1849083.917       344992.53     1847899.954      345320.787
     1847438.896       346370.61     1846436.441      345805.785
     1845038.429      347806.017     1843789.333       347640.63
     1843291.763      346954.227     1842168.116      346629.153
     1841674.074        347337.2     1839713.824      347455.775
     1837887.774       349294.94     1832578.795      348331.229
     1831221.634      349267.849     1829912.381       348328.26
     1828667.238      349688.091     1826800.724      347859.447
     1824994.179      348087.431     1825004.643      349692.095
     1823848.044      350062.032     1823349.222      351154.832
     1822062.368       351235.62     1820442.032      349594.533
     1819560.288      350986.913     1817870.541      350209.779
     1817353.873      350723.873     1817325.702      352527.378
     1815817.429      352565.191     1815091.402      353451.438

Type RM Length L Ch R = 1 ,51213.8 ,311.8,311.1,310.4
XS GIS Cut Line= 3
     1850993.774      343856.534     1851258.953      344333.814
     1851524.132      344811.094
#Sta/Elev= 30
       0 1343.52    39.7 1325.01    69.5 1313.17    79.4 1313.01   109.2 1298.88
   168.8 1264.11   188.6  1257.8   228.3 1231.57     268 1210.21   367.3 1176.86
   397.1    1162     417 1156.68   506.3 1120.84   528.5 1117.44   555.9 1117.39
   563.5 1118.28   595.6 1130.09   645.3 1138.68   694.9 1161.57   734.6 1187.89
   744.6 1191.06   804.1 1236.17   833.9 1254.07   863.7 1266.51   893.4 1285.58
   943.1 1322.95     963  1329.9  1062.2 1400.24  1072.2 1402.09    1092 1413.52
#Mann= 3 , 0 , 0
       0      .1       0   528.5    .045       0   563.5      .1       0
Bank Sta=528.5,563.5
XS Rating Curve= 0 ,0
Exp/Cntr=0.3,0.1

Type RM Length L Ch R = 1 ,50902.7 ,266,302.3,338.5
XS GIS Cut Line= 3
     1850908.968      343895.162     1850955.848      344431.442
     1851258.042      344949.869
#Sta/Elev= 30
       0 1296.64      10  1291.1    19.9 1290.57   109.7 1250.48   129.6 1246.36
   199.4 1209.78   209.4 1208.44   249.2 1193.72   289.1 1185.58   368.8 1181.59
   408.7 1168.29   488.5 1129.56   518.4 1126.32   548.3 1119.03   582.7 1117.41
   588.3  1117.4   617.7 1117.61   678.3 1127.62   708.4 1150.72   718.4 1151.02
   748.4 1176.25   818.4 1227.19   838.4 1233.92   938.4  1306.9   948.4 1308.62
   958.4 1314.68  1008.4 1349.26  1038.4 1373.36  1058.4 1382.59  1138.4 1451.09
#Mann= 3 , 0 , 0
       0      .1       0   582.7    .045       0   617.7      .1       0
Bank Sta=582.7,617.7
XS Rating Curve= 0 ,0
Exp/Cntr=0.3,0.1

Type RM Length L Ch R = 1 ,50600.4 ,287.6,286.6,283.5
XS GIS Cut Line= 3
     1850826.443      343897.154     1850745.481      344420.009
     1850407.098       344938.24
#Sta/Elev= 30
       0 1264.79    59.9 1246.64    99.8 1230.63   109.8 1230.06   199.7 1194.17
   269.5 1178.73   319.4 1174.19   389.3 1152.42   409.3 1148.88   479.2 1125.48
   519.1 1123.35     559 1113.75     596 1111.18   628.9 1110.37     631 1110.77
   638.9 1112.28   678.8 1129.35   698.8 1149.28   708.8 1156.76   718.8 1161.04
   768.7  1206.7   808.6 1238.54   828.6 1245.96   878.5 1282.18   898.4 1292.06
   968.3 1276.77  1028.2 1250.66  1098.1 1228.27    1128 1223.57    1148 1227.69
#Mann= 3 , 0 , 0
       0      .1       0     596    .045       0     631      .1       0
Bank Sta=596,631
XS Rating Curve= 0 ,0
Exp/Cntr=0.3,0.1

Type RM Length L Ch R = 1 ,50313.8 ,294.8,297.1,301.4
XS GIS Cut Line= 3
     1850750.289      343857.376     1850464.374      344326.594
     1850207.419      344814.516
#Sta/Elev= 30
       0 1242.74      50 1222.78   109.9 1207.38   129.9 1206.93   179.8 1199.29
   259.8  1172.7   269.7 1170.21   279.7 1169.82   349.7 1152.49   469.5 1120.27
     532 1109.67   549.5 1109.58   559.3 1110.16   588.9 1121.25   618.4 1124.47
   628.2 1128.17   657.8 1147.06   697.2 1160.69     707 1160.06   746.4 1168.27
     776 1171.04   805.5 1172.48     835 1168.87   874.4 1173.48   933.5 1188.47
     963 1198.22   982.8 1206.73  1012.3 1216.38    1032 1220.55  1100.9 1244.57
#Mann= 3 , 0 , 0
       0      .1       0     532    .045       0   559.3      .1       0
Bank Sta=532,559.3
XS Rating Curve= 0 ,0
Exp/Cntr=0.3,0.1

Type RM Length L Ch R = 1 ,50016.7 ,322.3,309.1,295.9
XS GIS Cut Line= 3
      1850532.96      343715.606       1850162.4      344239.368
     1850133.285      344775.971
#Sta/Elev= 30
       0 1315.23      79 1329.61   108.6 1326.72   118.4 1323.07   138.2 1309.66
   177.7 1273.66   207.3 1250.83     227 1244.31     306 1194.46   325.7 1183.97
   345.5 1179.44   424.4 1140.68     454 1131.02   503.4 1106.55   512.7 1106.15
   547.7  1106.1   572.5 1106.07   641.6 1122.38   731.2 1125.04     761 1138.59
     771 1139.55   830.7 1167.18   870.5 1172.41   900.3 1181.03   950.1 1202.81
     960 1203.14   989.9 1216.83  1019.8 1225.33  1099.4 1237.24    1179 1240.61
#Mann= 3 , 0 , 0
       0      .1       0   512.7    .045       0   547.7      .1       0
Bank Sta=512.7,547.7
XS Rating Curve= 0 ,0
Exp/Cntr=0.3,0.1

Type RM Length L Ch R = 1 ,49707.6 ,350.3,322.1,294
XS GIS Cut Line= 3
     1850068.448      343499.422     1849938.314      344099.886
      1850063.14      344753.247
#Sta/Elev= 30
       0 1422.07     9.9 1419.87    29.7 1409.33    99.1 1350.99     109 1351.13
   188.3 1287.86   208.1 1281.51   227.9 1267.16   247.7 1250.09   277.5 1219.91
   297.3 1209.95   346.8 1159.84   386.5  1128.1   396.4 1127.67     436 1112.08
   465.8 1106.61   485.6  1106.1   490.4  1106.1   525.4 1106.11     545    1108
   614.4 1125.81   783.2 1119.79   882.5 1125.69   961.9 1159.03   981.7 1163.18
  1051.2 1191.86  1071.1 1196.19  1140.6 1227.56  1210.1 1233.67  1279.6 1231.38
#Mann= 3 , 0 , 0
       0      .1       0   490.4    .045       0   525.4      .1       0
Bank Sta=490.4,525.4
XS Rating Curve= 0 ,0
Exp/Cntr=0.3,0.1

Type RM Length L Ch R = 1 ,49385.5 ,317.5,298.4,279.3
XS GIS Cut Line= 3
     1849363.095      343705.066      1849833.13      344323.972
     1849990.416      344776.597
#Sta/Elev= 30
       0  1415.3    39.8 1381.18    59.8 1367.02    79.7 1357.58   119.6 1328.78
   149.4 1305.94   169.4 1285.16   189.3 1269.38   209.2 1258.07   288.9 1180.31
   308.9  1156.4   318.8  1147.8   368.6  1124.1   398.5 1118.93   448.4 1105.28
   478.2  1102.8   494.4  1102.8   529.4  1102.8   577.9 1103.55   607.8  1114.2
   637.7 1119.18   757.2 1117.46     867 1125.64     897 1137.85   906.9 1138.53
   996.8 1179.86  1016.8 1184.63  1096.6 1221.06  1196.4 1215.05  1256.3  1214.7
#Mann= 3 , 0 , 0
       0      .1       0   494.4    .045       0   529.4      .1       0
Bank Sta=494.4,529.4
XS Rating Curve= 0 ,0
Exp/Cntr=0.3,0.1

Type RM Length L Ch R = 1 ,49087.1 ,255.8,253.5,251.2
XS GIS Cut Line= 3
     1848979.915      344147.306     1849737.094      344420.009
     1849928.419      344825.604
#Sta/Elev= 30
       0 1287.51    39.7  1298.8   109.3 1312.08   119.2 1316.77   208.6 1326.06
   238.5 1324.33   258.3 1312.96   278.2 1296.79   288.1 1281.23   357.7 1219.62
   377.6 1194.28   447.1 1138.69     457 1126.41   486.8 1104.98   503.9 1097.49
   536.5 1096.08   538.9 1096.11   556.4 1097.24     626 1117.24   735.2 1112.06
     775 1115.62   814.8 1123.18   884.5 1128.97   924.4 1147.07   934.3 1148.38
   994.1 1183.74    1034 1203.94  1063.9 1212.13  1193.4 1198.47  1253.2 1208.13
#Mann= 3 , 0 , 0
       0      .1       0   503.9    .045       0   538.9      .1       0
Bank Sta=503.9,538.9
XS Rating Curve= 0 ,0
Exp/Cntr=0.3,0.1

Type RM Length L Ch R = 1 ,48833.6 ,312.7,332.2,351.7
XS GIS Cut Line= 3
      1848878.39      344419.738     1849654.776      344639.522
     1849892.021      344895.885
#Sta/Elev= 30
       0  1192.8    19.9 1188.74    79.7 1188.83   219.2 1175.98   298.8 1179.19
   328.7  1193.4   348.7 1197.53   358.6 1194.26   388.5 1175.96   398.5 1164.98
   468.2 1123.67   488.1 1109.16     508 1100.24   520.7 1097.03   537.9 1096.09
   555.7 1096.31   597.7 1107.29   637.6 1108.72   697.3 1115.95   727.2 1122.02
     787 1128.23   796.9 1130.41   856.8 1165.16   886.7 1178.76   926.6  1186.1
   966.6 1183.28   986.5 1185.57  1046.4 1198.98  1096.3 1206.93  1156.2 1223.34
#Mann= 3 , 0 , 0
       0      .1       0   520.7    .045       0   555.7      .1       0
Bank Sta=520.7,555.7
XS Rating Curve= 0 ,0
Exp/Cntr=0.3,0.1

Type RM Length L Ch R = 1 ,48501.3 ,283.3,287.5,291.8
XS GIS Cut Line= 3
     1848836.038      344493.316     1849174.592      344737.845
       1849631.4      345265.933
#Sta/Elev= 30
       0 1197.79    29.8 1189.04    49.7 1179.66   109.4 1165.09   248.6 1148.17
   308.2 1144.27   328.1 1141.56     348 1136.96   367.9 1134.27   447.6 1114.21
   477.5 1109.17   517.4    1106   557.2 1097.59   577.2  1096.1   592.2 1097.46
   597.2 1098.67   627.1 1118.32     687 1121.02   696.9 1127.64   716.9 1150.62
   726.8 1156.85   746.8 1164.33   766.8 1167.86   876.5 1210.31   896.4 1213.18
   956.3  1236.3  1006.2 1251.59  1026.1 1252.97    1056 1260.24  1115.9 1271.19
#Mann= 3 , 0 , 0
       0      .1       0   557.2    .045       0   592.2      .1       0
Bank Sta=557.2,592.2
XS Rating Curve= 0 ,0
Exp/Cntr=0.3,0.1

Type RM Length L Ch R = 1 ,48213.8 ,295.6,300,297.9
XS GIS Cut Line= 3
     1848740.865      344564.697     1849041.262      345020.633
      1849341.66      345476.569
#Sta/Elev= 30
       0 1208.29    79.4 1212.31    99.3 1211.09     139 1203.38   198.6 1202.56
   228.3 1190.19   258.1 1174.61   327.6 1146.74   367.3 1135.12   397.1 1129.18
   496.4 1099.91   528.5 1096.13   536.1  1096.1   563.5  1096.1   585.7 1097.51
   615.5 1109.88   635.4  1114.7   665.1 1112.92     675 1114.48     685 1119.63
   694.9 1128.25   714.8 1150.09   724.7    1156   734.6  1158.4   843.8 1224.34
   913.3 1261.78     963 1294.66   982.8 1298.93  1002.6 1315.84    1092  1383.2
#Mann= 3 , 0 , 0
       0      .1       0   528.5    .045       0   563.5      .1       0
Bank Sta=528.5,563.5
XS Rating Curve= 0 ,0
Exp/Cntr=0.3,0.1

Type RM Length L Ch R = 1 ,47913.8 ,290.1,300,315.8
XS GIS Cut Line= 3
     1848550.341      344687.949     1848792.144      345187.548
      1849120.34      345621.903
#Sta/Elev= 30
       0 1167.27    29.7 1156.88    49.6 1154.22   138.8  1162.9     218 1157.49
   307.2 1135.42   327.1 1133.08   396.5 1114.46   455.9 1105.02   495.6 1102.26
   515.4 1097.07   537.5 1096.12   545.1  1096.1   572.5  1096.1   594.6 1098.71
   624.3 1110.65     654 1112.83   693.6  1129.5   713.4 1142.26   733.2 1158.93
   762.9 1195.62   772.8 1203.27   792.6 1210.18     852 1266.82   891.6 1312.19
   901.5 1315.34     951 1341.56  1020.3 1382.38  1030.2 1379.85  1099.4 1402.91
#Mann= 3 , 0 , 0
       0      .1       0   537.5    .045       0   572.5      .1       0
Bank Sta=537.5,572.5
XS Rating Curve= 0 ,0
Exp/Cntr=0.3,0.1

Type RM Length L Ch R = 1 ,47613.8 ,202.8,206.2,209.8
XS GIS Cut Line= 3
     1848423.149      344715.233     1848502.594      345255.364
     1848591.643      345794.382
#Sta/Elev= 30
       0 1179.29    49.6 1168.07    69.5 1165.79     129 1154.03   258.1 1137.69
   337.5 1122.79   347.4 1122.47   436.8 1106.84   446.7 1106.77   476.5 1099.47
   528.4 1090.26   545.9    1090   563.4 1091.06   605.5 1105.04   665.1 1109.99
     685 1114.69   704.9 1125.65   734.7 1151.21   744.6 1156.38   754.5 1158.51
   764.5  1163.6   794.3 1173.58   824.1  1180.3   863.8 1186.61   903.5 1198.05
   933.3 1204.64   943.3 1205.09  1022.7 1224.16  1042.6 1227.24  1092.3 1241.04
#Mann= 3 , 0 , 0
       0      .1       0   528.4    .045       0   563.4      .1       0
Bank Sta=528.4,563.4
XS Rating Curve= 0 ,0
Exp/Cntr=0.3,0.1

Type RM Length L Ch R = 1 ,47407.6 ,589,552.6,516.7
XS GIS Cut Line= 3
     1848272.081      344746.105     1848310.259      345366.658
     1848490.463      345828.054
#Sta/Elev= 30
       0 1178.04   128.3 1163.85   177.6 1153.68   217.1 1149.76   315.8 1134.28
   394.8 1116.27   404.6 1115.27   434.2 1102.48     454 1097.38   473.7 1096.65
     523 1097.95   551.4 1090.52   562.5    1090   586.4 1090.19   592.1  1090.2
   621.7 1100.44   671.3 1102.82   681.2 1104.61     701 1114.71   710.9 1116.53
   720.8 1121.94   760.4 1136.83     800 1148.84   819.9 1151.74   889.2 1167.97
   978.4 1182.66  1008.1 1190.84  1027.9 1194.08  1107.2 1213.03  1117.1 1214.05
#Mann= 3 , 0 , 0
       0      .1       0   551.4    .045       0   586.4      .1       0
Bank Sta=551.4,586.4
XS Rating Curve= 0 ,0
Exp/Cntr=0.3,0.1

Type RM Length L Ch R = 1 ,46854.9 ,192.8,190.6,188.5
XS GIS Cut Line= 3
     1847539.677      345307.207     1848118.185      345563.305
     1848329.817      345864.126
#Sta/Elev= 30
       0 1238.54    59.3 1238.66   128.5 1227.44   138.4 1224.87   158.2 1216.69
     168 1210.09   177.9 1201.43   207.6 1170.41   217.5 1150.43   227.4 1136.71
     257 1103.23   266.9 1093.52   276.8 1087.45   286.7 1085.75   316.7 1085.97
   351.7 1085.79   365.8 1085.56   385.5 1086.82   395.4 1090.06   425.1 1092.37
   484.4  1095.1   553.6 1095.28   632.7 1100.38   692.3 1117.77   712.2 1120.65
   791.7 1138.82   821.5 1146.98   841.4  1149.8   950.8 1172.25  1000.5 1180.91
#Mann= 3 , 0 , 0
       0      .1       0   316.7    .045       0   351.7      .1       0
Bank Sta=316.7,351.7
XS Rating Curve= 0 ,0
Exp/Cntr=0.3,0.1

Type RM Length L Ch R = 1 ,46664.2 ,350.6,347.2,343.9
XS GIS Cut Line= 3
     1847361.375      345188.836     1847596.842      345554.159
     1848221.082      345782.818
#Sta/Elev= 30
       0 1287.47     9.9 1283.13    19.8  1283.3    29.6 1280.03   128.4 1235.58
   167.9 1229.94   207.4 1230.57   256.8 1225.09   276.6  1214.3   296.3 1209.91
   365.5 1201.69     405 1186.88   424.8 1170.97   434.6 1166.96   504.1 1117.22
     514 1106.18   523.9  1101.4   563.6 1087.52   623.2 1082.04   658.2  1081.9
   672.8 1081.83   702.5 1092.62   712.5 1094.08   821.6 1095.05     901 1098.64
   930.8 1109.66   980.4 1117.18  1000.2 1122.96    1020 1132.36  1099.4 1153.12
#Mann= 3 , 0 , 0
       0      .1       0   623.2    .045       0   658.2      .1       0
Bank Sta=623.2,658.2
XS Rating Curve= 0 ,0
Exp/Cntr=0.3,0.1

Type RM Length L Ch R = 1 ,46317   ,479.4,519.5,559.5
XS GIS Cut Line= 3
      1847363.61      345316.353     1847560.257      345924.587
     1848183.114      346082.891
#Sta/Elev= 30
       0 1270.75    49.9 1282.92   159.8 1290.66   169.8 1289.85   189.8 1282.84
   199.8  1282.8   239.7 1264.88   279.7 1243.32   309.6 1232.45   389.5 1183.38
   399.5 1182.96   429.5 1167.61   489.4 1145.02   549.3 1135.33   559.3 1128.41
   589.3 1097.33   649.1 1089.16     748 1084.82   773.3 1079.54   787.5 1078.59
   808.3 1078.85   846.9 1086.74   916.1  1086.1   995.2  1090.8  1034.7 1099.06
  1074.3  1104.3  1153.4 1125.49    1183 1138.22  1222.6 1142.52  1281.9 1166.98
#Mann= 3 , 0 , 0
       0      .1       0   773.3    .045       0   808.3      .1       0
Bank Sta=773.3,808.3
XS Rating Curve= 0 ,0
Exp/Cntr=0.3,0.1

Type RM Length L Ch R = 1 ,45797.6 ,224.4,257.9,291.3
XS GIS Cut Line= 3
     1847404.768      345691.355     1847411.628       346265.29
     1847466.506      346761.099
#Sta/Elev= 30
       0 1175.39     9.9 1173.24    79.2 1130.78    89.1 1126.84      99  1125.7
   128.6 1111.07   158.3 1094.98   168.2 1091.16   178.1 1090.57   197.9 1092.24
   217.7 1096.27   227.6 1094.34   247.4 1087.52   257.3 1086.62   484.9 1083.16
   564.1 1079.95   663.8 1077.84   693.7 1073.83   703.7  1073.7   713.6 1073.92
   723.6  1075.9   743.6 1084.48   753.6 1087.57   773.5 1090.68   823.4 1112.12
   843.4 1117.92   893.2 1127.14   913.2 1128.64   963.1  1127.6  1072.8  1120.6
#Mann= 3 , 0 , 0
       0      .1       0   693.7    .045       0   713.6      .1       0
Bank Sta=693.7,713.6
XS Rating Curve= 0 ,0
Exp/Cntr=0.3,0.1

Type RM Length L Ch R = 1 ,45539.7 ,232.2,230.4,228.6
XS GIS Cut Line= 3
     1847378.091      345663.534     1847307.969      346218.414
      1846824.54      346606.421
#Sta/Elev= 30
       0 1187.52      20  1174.5      40 1167.73   109.9 1123.03   129.8 1116.42
   169.8  1093.7   179.8 1089.88   189.8 1088.87   209.7 1091.08   219.7 1090.36
   249.7 1084.64   339.6 1085.33   679.3 1076.67   689.3 1075.42   709.3 1070.03
   729.3  1069.5   739.3 1069.73   749.3 1070.96   769.2 1076.27   779.2 1080.48
   789.2 1088.55   819.2  1122.6   829.2 1131.54   889.2 1153.55   939.2 1169.38
   959.2 1179.76  1029.2 1204.12  1039.2 1205.78  1109.2 1206.26  1179.2 1199.33
#Mann= 3 , 0 , 0
       0      .1       0   709.3    .045       0   739.3      .1       0
Bank Sta=709.3,739.3
XS Rating Curve= 0 ,0
Exp/Cntr=0.3,0.1

Type RM Length L Ch R = 1 ,45309.3 ,149.3,143.8,138.2
XS GIS Cut Line= 3
     1847352.177      345691.355      1847249.28      345954.313
     1846698.211      346448.217
#Sta/Elev= 30
       0 1166.06     9.7 1163.75    87.6  1114.2   107.1 1107.95   136.3 1091.13
   155.8 1089.38     185 1082.81   194.7 1082.17   282.4 1080.72   432.4 1075.28
   482.4 1075.92   492.4 1075.03   509.3 1068.04   522.4 1064.17   532.4 1064.13
   544.3 1065.89   562.4 1072.55   582.4 1074.62   592.4 1077.43   602.4 1085.28
   622.4 1106.55   632.4 1115.58   672.4 1126.26   702.4 1133.31   722.4  1134.6
   842.4 1161.57   862.4 1161.95   932.4 1175.85   972.4  1179.6  1022.4 1178.71
#Mann= 3 , 0 , 0
       0      .1       0   509.3    .045       0   544.3      .1       0
Bank Sta=509.3,544.3
XS Rating Curve= 0 ,0
Exp/Cntr=0.3,0.1

Type RM Length L Ch R = 1 ,45165.5 ,532.6,501.7,470.8
XS GIS Cut Line= 3
     1847137.237      345341.506     1847153.243      345791.965
     1846693.638      346363.613
#Sta/Elev= 30
       0 1344.77    19.6 1327.35    29.4 1321.27    58.8 1309.51   137.2 1238.23
     147 1231.19   156.8 1230.91     196 1201.31   235.2 1174.79     245 1174.04
   313.6 1133.41   333.2 1123.04   352.8 1117.99   401.8 1090.81   460.7  1076.5
   609.3 1070.85   668.8 1073.23   697.1 1067.17   718.4 1064.09   732.1 1065.36
     758 1072.26   827.4 1074.46     867 1090.12   896.8 1099.28   906.7 1099.44
  1005.8 1125.48  1025.6 1127.03  1134.7 1154.63  1154.5 1155.98  1184.2 1162.74
#Mann= 3 , 0 , 0
       0     .06       0   697.1    .045       0   732.1     .06       0
Bank Sta=697.1,732.1
XS Rating Curve= 0 ,0
Exp/Cntr=0.3,0.1

Type RM Length L Ch R = 1 ,44663.8 ,407.4,394.6,381.8
XS GIS Cut Line= 3
     1846526.716      345250.042     1846764.522      346102.941
     1846597.775      346529.862
#Sta/Elev= 30
       0  1317.9      10 1312.83    19.9 1312.46    49.7 1295.71   109.4 1269.88
   129.3 1270.41   139.3 1266.58   159.2 1251.74     189 1225.43   218.9 1203.26
   228.8 1197.53   238.8 1196.29   318.4  1114.2   328.3 1113.43   348.2  1096.2
   368.1 1085.32   443.6 1065.14   467.6 1063.63   478.6 1063.76   517.3 1071.56
   646.7 1070.47   855.6 1075.86   915.3 1093.61   935.2 1096.24    1015 1119.82
  1034.9 1122.35  1114.6 1146.35  1134.5 1148.94  1204.3 1171.29  1343.8 1179.12
#Mann= 3 , 0 , 0
       0     .06       0   443.6    .045       0   478.6     .06       0
Bank Sta=443.6,478.6
XS Rating Curve= 0 ,0
Exp/Cntr=0.3,0.1

Type RM Length L Ch R = 1 ,44269.2 ,263.9,258.6,253.4
XS GIS Cut Line= 3
     1846000.728      345498.507     1846529.003      346166.966
     1846530.179      346558.082
#Sta/Elev= 30
       0 1405.14    49.5 1366.58    69.4 1356.41    89.2 1344.05   178.3 1279.33
   277.4 1216.03   336.8 1173.08   396.3    1136   435.9 1102.88   445.8 1090.91
   455.7 1081.79   465.6 1076.47   475.5 1075.35   485.4  1071.9   508.7 1059.68
   515.2 1057.19   525.1 1056.22   543.7 1056.88   594.4 1064.78   792.6 1066.88
   871.6 1070.37   881.3  1072.3   900.9 1079.68   920.4 1083.72   998.7  1119.8
  1018.2 1124.23  1096.4 1157.18  1125.8 1163.53  1174.7 1169.19  1243.1 1172.82
#Mann= 3 , 0 , 0
       0     .06       0   508.7    .045       0   543.7     .06       0
Bank Sta=508.7,543.7
XS Rating Curve= 0 ,0
Exp/Cntr=0.3,0.1

Type RM Length L Ch R = 1 ,44010.5 ,367.1,365.1,363.1
XS GIS Cut Line= 3
     1845763.541        345742.5     1846364.368      346297.302
     1846469.075      346606.023
#Sta/Elev= 30
       0 1274.26    59.8 1270.22    79.8 1271.89   109.7 1268.44   129.6 1271.82
   169.5 1263.61   199.5 1239.16   239.4 1211.48   259.3 1198.85   279.2 1192.37
   319.1 1164.74     389 1122.92   398.9  1113.9   408.9 1107.55   428.8  1099.1
   458.8 1080.47   488.7 1067.72   508.6 1053.63   521.2 1051.61   538.6 1051.49
   556.2 1054.05   588.4 1061.28   618.3 1063.66   807.8 1067.46   837.6 1076.98
   936.3 1134.24   946.2 1135.18   975.9 1151.73  1084.5 1155.48  1143.8 1165.12
#Mann= 3 , 0 , 0
       0     .06       0   521.2    .045       0   556.2     .06       0
Bank Sta=521.2,556.2
XS Rating Curve= 0 ,0
Exp/Cntr=0.3,0.1

Type RM Length L Ch R = 1 ,43645.4 ,232.6,231.6,230.6
XS GIS Cut Line= 3
     1845521.118      346058.406     1845944.202      346403.537
     1846367.287      346748.668
#Sta/Elev= 30
       0 1225.31    69.5 1200.44    89.4 1190.61    99.3 1181.71   109.2 1177.68
     139 1167.82   188.6 1154.04   208.5 1146.73   317.7 1142.82   337.5  1139.9
   347.4 1136.68   367.3 1127.16   377.2 1124.15   387.2 1117.74   397.1    1110
     407 1096.86     417  1087.4   436.8 1073.01   486.4 1053.54   506.3 1051.59
   511.1 1051.63   546.1 1053.84   575.8 1057.03     814  1066.4     824 1067.98
   853.8 1081.02   923.2 1119.39   933.2 1120.93   992.7 1118.44    1092 1131.89
#Mann= 3 , 0 , 0
       0     .06       0   511.1    .045       0   546.1     .06       0
Bank Sta=511.1,546.1
XS Rating Curve= 0 ,0
Exp/Cntr=0.3,0.1

Type RM Length L Ch R = 1 ,43413.8 ,180.4,178.2,175.9
XS GIS Cut Line= 3
     1845358.055       346245.65      1845791.59      346577.558
     1846225.125      346909.466
#Sta/Elev= 30
       0 1375.52     9.9 1370.72    29.8 1352.95    49.6 1342.02   109.2 1313.36
     129 1293.47   188.6 1250.41   218.4 1230.89   228.3 1219.78   307.8 1171.24
   317.7 1164.78   327.6 1154.58     417 1098.95   426.9 1087.97   446.7 1073.37
   456.6 1067.82   506.3 1053.36   526.2  1051.6   528.5  1051.6   563.5 1051.97
   615.5  1056.2   714.8 1060.07   873.6 1060.67   903.4 1062.66     953 1069.11
   972.9 1073.65  1002.6 1090.41  1022.5 1106.52  1072.2  1129.2    1092 1135.16
#Mann= 3 , 0 , 0
       0     .06       0   528.5    .045       0   563.5     .06       0
Bank Sta=528.5,563.5
XS Rating Curve= 0 ,0
Exp/Cntr=0.3,0.1

Type RM Length L Ch R = 1 ,43235.6 ,424.6,421.8,419.9
XS GIS Cut Line= 3
     1845215.807      346409.765     1845671.164      346711.039
     1846126.521      347012.313
#Sta/Elev= 30
       0 1350.74    19.8 1351.06    59.6 1343.76    89.4  1336.2    99.3 1336.28
   109.2 1333.37     139  1317.9   188.6 1286.64   208.5 1268.47   238.2    1248
     268 1228.55   287.9  1218.6   307.8 1198.15   387.2 1140.34   397.1 1128.16
   446.7 1091.01   466.6  1080.1   476.5 1072.02   486.4 1066.31   526.2 1052.57
   543.3 1048.81   565.8  1048.4   578.3 1048.69   615.5 1053.27     963 1062.85
   972.9 1065.81  1012.6 1084.33  1042.4 1099.78  1062.2 1114.09    1092  1127.7
#Mann= 3 , 0 , 0
       0     .06       0   543.3    .045       0   578.3     .06       0
Bank Sta=543.3,578.3
XS Rating Curve= 0 ,0
Exp/Cntr=0.3,0.1

Type RM Length L Ch R = 1 ,42813.8 ,457.4,462.1,465.9
XS GIS Cut Line= 3
     1844971.545      346809.986     1845450.999      347071.104
      1845987.08      347381.147
#Sta/Elev= 30
       0 1166.33    39.7 1163.34    59.6 1164.95    89.3 1161.61   119.1 1155.75
     139 1150.55   208.4 1136.91   228.3 1131.23   248.2 1127.02   297.8 1117.54
   317.6 1111.94   387.1 1096.79     397 1094.16     407 1089.89   436.8 1084.37
   486.4 1061.05   506.2 1055.57   516.2 1051.29   528.4  1048.8     536 1048.49
   563.4 1048.78   685.8 1054.21  1005.4 1059.11  1085.3 1063.55  1095.3  1065.4
  1105.3 1068.71  1115.3 1073.44  1125.3 1079.97  1135.3 1088.02  1165.2  1103.6
#Mann= 3 , 0 , 0
       0     .06       0   528.4    .045       0   563.4     .06       0
Bank Sta=528.4,563.4
XS Rating Curve= 0 ,0
Exp/Cntr=0.3,0.1

Type RM Length L Ch R = 1 ,42351.6 ,128.3,133.7,139.1
XS GIS Cut Line= 3
     1845001.559       347298.83     1845436.011      347618.953
     1845568.634      347845.326
#Sta/Elev= 30
       0 1104.48      50 1104.37    99.9 1106.24   109.9 1105.32   119.9 1102.67
   149.9 1072.52   159.9 1063.39   169.9 1056.26   229.8 1050.47   239.8  1048.9
   259.8 1044.18   269.8 1043.04   279.8  1042.9   319.8 1042.94   369.8 1049.36
   489.7 1056.16   499.7 1057.06   539.7 1061.36   559.1 1062.67     598 1067.03
   627.1 1070.81   646.5 1073.99   656.3 1073.87     666 1076.27   685.4 1082.36
   724.3 1096.16     734 1098.66   763.2 1104.09   772.9 1105.44     802 1111.73
#Mann= 3 , 0 , 0
       0     .06       0   269.8    .045       0   319.8     .06       0
Bank Sta=269.8,319.8
XS Rating Curve= 0 ,0
Exp/Cntr=0.3,0.1

Type RM Length L Ch R = 1 ,42218   ,254.1,275.6,297
XS GIS Cut Line= 4
     1845012.992      347358.281     1845027.829      347432.543
     1845323.968      347735.569     1845415.432      347971.088
#Sta/Elev= 30
       0 1097.95    18.9 1097.01    28.4 1093.42    37.9 1086.89    56.8 1079.81
    75.7 1064.29    85.6    1057    95.4 1053.98   105.3 1053.18   184.1 1050.77
   243.2 1047.39   282.6 1043.16   302.4  1042.9   304.7  1042.9   339.7 1043.44
   381.2 1050.54     460 1055.88   509.2 1060.41   518.9 1062.03   528.6 1065.39
   567.4 1085.13   577.2 1086.47   586.9 1090.94   606.3  1102.1   635.5 1122.21
   674.4 1152.16   684.1 1153.55   693.8 1159.47   732.6 1191.28   752.1 1204.73
#Mann= 3 , 0 , 0
       0      .1       0   304.7    .045       0   339.7      .1       0
Bank Sta=304.7,339.7
XS Rating Curve= 0 ,0
Exp/Cntr=0.3,0.1

Type RM Length L Ch R = 1 ,41942.4 ,284.4,295.2,306
XS GIS Cut Line= 3
     1844978.693      347374.287     1844980.979      347454.318
     1845079.926      348328.608
#Sta/Elev= 30
       0 1091.04      10 1090.07      40 1081.72    70.1 1058.91    80.1 1053.94
    90.1 1052.33     390 1047.35     400 1046.23   419.5 1040.79     450 1040.35
   454.5 1040.54     470 1043.26     480 1047.71     510  1068.5     520 1070.05
     590 1129.91     610 1142.51     620 1143.28     640 1157.78     690 1207.27
     700 1215.52     710 1216.32     760 1252.77     780 1270.43     800 1291.83
     810 1293.16     850  1328.2   889.9 1359.57   909.9 1367.66   959.9 1403.78
#Mann= 3 , 0 , 0
       0      .1       0   419.5    .045       0   454.5      .1       0
Bank Sta=419.5,454.5
XS Rating Curve= 0 ,0
Exp/Cntr=0.3,0.1

Type RM Length L Ch R = 1 ,41647.2 ,188.2,191,193.8
XS GIS Cut Line= 3
     1844955.827      347022.152     1844816.345      347394.867
     1844633.417      348222.614
#Sta/Elev= 30
       0 1131.63    89.5 1118.27   278.6 1097.38   328.3 1086.08   358.2 1076.11
     388  1062.7   427.9  1051.5   467.8  1051.2   567.5 1045.23     757 1044.53
     767 1043.21   777.9 1039.52   796.9  1037.5   812.9 1038.81   836.8 1046.01
   866.7 1047.54   876.7 1051.02   886.6 1057.08   896.6  1059.3   936.5 1100.42
   986.4 1141.61   996.4 1141.84  1076.1 1204.79  1086.1 1206.96  1096.1 1212.21
    1146  1248.5  1155.9 1252.48  1165.9 1251.54  1185.8 1246.47  1245.7 1221.49
#Mann= 3 , 0 , 0
       0      .1       0   777.9    .045       0   812.9      .1       0
Bank Sta=777.9,812.9
XS Rating Curve= 0 ,0
Exp/Cntr=0.3,0.1

Type RM Length L Ch R = 1 ,41456.2 ,289.9,288.8,287.7
XS GIS Cut Line= 3
      1844769.43      347015.613     1844607.665      347537.104
     1844444.171       348058.05
#Sta/Elev= 30
       0  1104.6    59.6  1094.2   168.8 1082.74   198.6 1077.94   238.3 1070.08
   287.9 1055.17   297.8 1054.09   317.7  1047.5   327.6 1046.18     417 1049.45
     546 1045.16     685 1043.91   704.8 1042.69   714.8 1039.28   731.3 1037.57
   734.6  1037.5   744.6 1037.72   766.3 1043.14   784.3 1044.63   863.7  1046.1
   873.6 1049.85   883.5 1056.25   893.5 1056.43   943.1  1088.8   982.8 1105.18
  1002.7 1107.76  1032.4 1118.17  1042.4 1120.31  1082.1 1126.79    1092 1124.47
#Mann= 3 , 0 , 0
       0      .1       0   731.3    .045       0   766.3      .1       0
#XS Ineff= 2 , 0
          416.14 1049.82
Permanent Ineff=
       F       F
Bank Sta=731.3,766.3
XS Rating Curve= 0 ,0
Exp/Cntr=0.3,0.1

Type RM Length L Ch R = 1 ,41167.5 ,449.4,454.1,458.8
XS GIS Cut Line= 2
     1844489.362      346857.517      1844121.22      348186.028
#Sta/Elev= 30
       0 1120.96    59.9 1104.42   139.9 1070.18   149.8 1066.75   159.8 1065.04
   199.8 1046.37   219.8 1039.82   269.7 1039.42   419.6 1046.02   529.4  1040.8
   769.2 1040.91   799.2 1037.74   803.2 1037.74   838.2 1037.97     919 1043.33
    1009  1046.3    1019 1048.78  1028.9  1053.8  1038.9 1054.49  1078.9 1075.46
  1108.8  1089.4  1128.8 1096.82  1158.8 1101.93  1198.8 1104.25  1238.7 1112.35
  1318.6    1137  1328.6 1138.85  1338.6 1142.57  1358.6 1153.21  1378.6 1167.67
#Mann= 3 , 0 , 0
       0      .1       0   803.2    .045       0   838.2      .1       0
#XS Ineff= 2 , 0
          419.45 1046.02
Permanent Ineff=
       F       F
Bank Sta=803.2,838.2
XS Rating Curve= 0 ,0
Exp/Cntr=0.3,0.1

Type RM Length L Ch R = 1 ,40713.4 ,270.4,287.5,304.6
XS GIS Cut Line= 3
     1844246.983      346626.571     1843791.951      347703.557
      1843789.04      348176.521
#Sta/Elev= 30
       0  1161.8      50 1134.08    79.9 1121.29    89.9 1120.27   179.9 1077.35
   199.9 1072.22   269.8 1042.79   289.8 1037.66   409.7 1038.38   529.6 1042.45
  1049.2 1037.28  1085.1 1031.64  1089.2 1031.39  1120.1  1031.5  1139.2 1034.43
  1159.2 1042.37  1198.7 1070.68  1218.4 1077.81  1297.3 1134.28  1307.1 1138.92
    1317 1139.76  1336.7 1149.74  1356.4 1157.08    1386 1159.02  1425.4 1158.58
  1474.6 1150.57    1514 1148.41  1553.5 1158.54  1602.7 1168.32  1642.1  1184.3
#Mann= 3 , 0 , 0
       0      .1       0  1085.1    .045       0  1120.1      .1       0
#XS Ineff= 2 , 0
          519.79 1042.36
Permanent Ineff=
       F       F
Bank Sta=1085.1,1120.1
XS Rating Curve= 0 ,0
Exp/Cntr=0.3,0.1

Type RM Length L Ch R = 1 ,40425.9 ,264.4,267.3,270.2
XS GIS Cut Line= 3
     1844096.068      346779.773     1843860.548       347278.25
     1843153.082      347806.705
#Sta/Elev= 30
       0 1065.63     9.8  1061.5    19.7 1060.78    39.4 1053.65    68.9  1040.5
    78.8 1036.97    88.6 1035.37     315 1041.88   640.6 1038.54   878.7 1030.71
   879.9 1030.71   888.7 1030.74   914.9 1035.34   948.2 1039.97   987.9 1039.88
  1017.6 1041.59  1037.5  1048.4  1057.3 1051.23    1097 1061.47  1106.9 1064.83
  1116.9  1070.6  1126.8 1073.41  1186.3 1087.62  1206.2 1094.23  1216.1 1099.29
  1235.9 1105.68  1285.5 1117.04  1345.1  1122.3  1404.6  1115.1  1434.4 1123.74
#Mann= 3 , 0 , 0
       0      .1       0   879.9    .045       0   914.9      .1       0
#XS Ineff= 2 , 0
          305.48 1041.96
Permanent Ineff=
       F       F
Bank Sta=879.9,914.9
XS Rating Curve= 0 ,0
Exp/Cntr=0.3,0.1

Type RM Length L Ch R = 1 ,40158.4 ,365.1,344.7,324.4
XS GIS Cut Line= 4
     1844052.622      346626.571     1843808.589      347034.612
     1843245.455      347381.147     1843112.832      347712.703
#Sta/Elev= 30
       0 1125.36    19.8 1116.68    79.2 1087.01      99  1082.1   128.8 1066.25
   188.2 1038.86     208 1035.61   227.8 1034.79   435.8  1041.8   524.8 1038.49
   820.9  1032.5   872.8 1026.79   899.8  1026.4   907.8 1026.43   919.6  1027.2
   939.3 1031.18     959 1033.41  1087.3 1038.04  1126.8 1038.34  1176.3 1048.48
  1196.2 1051.08  1285.4 1070.18  1295.4  1071.2  1325.1 1080.52    1345  1084.9
  1374.7 1089.01  1414.4 1092.56  1434.2 1096.24  1454.1 1102.51  1493.8 1118.23
#Mann= 3 , 0 , 0
       0      .1       0   872.8    .045       0   907.8      .1       0
#XS Ineff= 2 , 0
          430.12  1041.8
Permanent Ineff=
       F       F
Bank Sta=872.8,907.8
XS Rating Curve= 0 ,0
Exp/Cntr=0.3,0.1

Type RM Length L Ch R = 1 ,39813.8 ,448,442.3,441.7
XS GIS Cut Line= 3
     1843467.254       346466.51      1843382.65      346747.761
     1843002.897      347625.992
#Sta/Elev= 30
       0 1097.28     9.8 1093.97    29.4 1091.78    68.5 1081.31    97.9 1075.45
   117.5 1069.64   127.3 1069.79   166.4 1057.76   205.6 1049.72   293.7 1040.19
   463.1 1032.64   502.3 1026.76   532.9 1026.45   537.3 1026.75   572.8 1031.32
   881.8 1036.43   931.6 1039.22   981.4 1058.31  1001.4 1064.23  1021.3 1067.72
  1041.2  1068.6    1101 1079.73    1121 1084.55  1140.9 1087.33  1180.8 1098.23
  1200.7 1102.38  1210.6 1102.88  1230.6 1111.28  1240.6 1112.61  1250.5 1115.95
#Mann= 3 , 0 , 0
       0      .1       0   502.3    .045       0   537.3      .1       0
Bank Sta=502.3,537.3
XS Rating Curve= 0 ,0
Exp/Cntr=0.3,0.1

Type RM Length L Ch R = 1 ,39371.5 ,191,196.3,196.9
XS GIS Cut Line= 3
     1843371.217      346537.394     1842984.783      346887.243
     1842698.959      347580.081
#Sta/Elev= 30
       0 1088.45    39.3 1079.39    49.2 1077.67      59 1077.66    98.4 1069.25
   127.9 1061.67     177 1046.63   196.7  1043.1   206.5  1039.5   255.7 1034.11
   304.9 1031.57   344.2  1032.7   432.8 1031.38   531.3 1033.07   591.2 1030.55
     705 1023.05   711.1    1023   731.1  1023.8     740 1025.83   761.1 1031.27
   781.1 1032.86     991 1031.41  1030.9 1033.21  1110.9 1040.52  1120.9 1042.86
  1180.8 1065.48  1200.8 1069.37  1210.8 1073.79  1230.8 1085.74  1270.8 1118.27
#Mann= 3 , 0 , 0
       0      .1       0     705    .045       0     740      .1       0
#XS Ineff= 2 , 0
                          811.03         1033.43
Permanent Ineff=
       F       F
Bank Sta=705,740
XS Rating Curve= 0 ,0
Exp/Cntr=0.3,0.1

Type RM Length L Ch R = 1 ,39175.2 ,260.2,264.8,258
XS GIS Cut Line= 3
     1843048.808       346345.32     1842936.765      346555.687
     1842553.887      347485.335
#Sta/Elev= 30
       0  1122.3    19.9 1107.32    29.8 1102.26    39.7 1099.44    69.5 1078.84
    79.4 1072.87    89.4 1068.58   129.1 1057.06     139 1055.92   158.9 1049.65
   198.6 1039.01   228.4 1031.42   238.3 1029.86   288.1  1028.3   397.6 1028.88
   596.7 1027.09   606.7 1026.56   626.6 1023.33   636.5 1022.98   642.1 1022.99
   677.1 1023.01   696.2 1024.04   736.1 1029.52   785.8 1031.69   994.9 1030.35
  1064.6 1031.04  1114.3 1033.19  1134.2 1035.44  1164.1 1040.55  1243.8 1074.22
#Mann= 3 , 0 , 0
       0      .1       0   642.1    .045       0   677.1      .1       0
#XS Ineff= 2 , 0
                          815.95         1031.77
Permanent Ineff=
       F       F
Bank Sta=642.1,677.1
XS Rating Curve= 0 ,0
Exp/Cntr=0.3,0.1

Type RM Length L Ch R = 1 ,38910.4 ,298.8,298.9,310.1
XS GIS Cut Line= 3
     1842823.283      346395.084     1842518.234      346904.654
      1842461.39      347455.627
#Sta/Elev= 30
       0 1039.87    19.8 1037.99    89.1 1035.13   108.9 1031.82   118.8 1031.28
   148.5 1031.38     198 1030.46     386 1025.74   514.7 1023.37   524.6 1022.45
   544.4  1019.3   554.3  1018.9   564.5 1018.92   574.1  1019.4   593.9 1026.58
   599.5 1027.59   603.8 1028.37   633.5 1028.91   712.6 1027.34   870.8 1025.77
   910.4 1026.18   989.5 1029.17    1039 1030.41  1048.9 1032.67  1078.6 1045.33
  1088.4 1046.44  1098.3  1049.3  1118.1  1057.8    1128 1062.63  1147.8 1073.54
#Mann= 3 , 0 , 0
       0      .1       0   564.5    .045       0   599.5      .1       0
#XS Ineff= 2 , 0
                          633.56          1028.9
Permanent Ineff=
       F       F
Bank Sta=564.5,599.5
XS Rating Curve= 0 ,0
Exp/Cntr=0.3,0.1

Type RM Length L Ch R = 1 ,38611.5 ,629.6,572.9,515
XS GIS Cut Line= 3
     1842967.204       345616.67     1842301.092      346715.748
     1842333.104      347436.025
#Sta/Elev= 30
       0 1225.94    19.9 1220.18    59.8 1216.14   109.6 1216.03   179.3 1232.33
   209.2 1236.41     269 1232.97   298.9 1226.29   368.6  1197.1   418.4 1163.91
   438.4 1155.32   468.2 1126.86     528  1079.1     538 1076.93   597.8 1044.83
   617.7 1040.44   836.9 1033.56   906.6 1027.55  1195.5 1026.82  1217.5 1017.92
  1235.4  1016.4  1252.5 1016.78  1285.2 1021.76  1413.6 1024.21  1848.1 1023.63
  1867.9 1027.03  1897.5 1039.61  1956.8 1070.84  1976.5 1076.24  2006.2 1095.36
#Mann= 3 , 0 , 0
       0      .1       0  1217.5    .045       0  1252.5      .1       0
Bank Sta=1217.5,1252.5
XS Rating Curve= 0 ,0
Exp/Cntr=0.3,0.1

Type RM Length L Ch R = 1 ,38038.5 ,317.2,330.1,343.1
XS GIS Cut Line= 5
     1841238.668      345796.258     1841364.595      346489.759
     1841846.861      346903.844     1842111.305      347029.012
     1842295.396      347494.352
#Sta/Elev= 30
       0 1228.94    49.6 1210.68   119.1 1176.98     139 1172.13   178.7    1154
   218.4  1130.8   258.1 1116.55     278 1114.69   317.7 1120.02   347.5 1119.81
     417 1094.87   506.3 1070.88   526.2  1067.6   605.6 1041.45   655.2 1038.26
   704.8 1029.51   843.9 1024.59    1261 1021.95    1399 1018.26  1450.9 1012.46
  1467.3 1012.36  1485.9 1012.96    1516 1017.72  1883.3 1020.58  1913.3 1033.74
  1923.3 1033.63  2003.4 1079.07  2023.4 1083.94  2113.5 1144.37  2133.5 1149.42
#Mann= 3 , 0 , 0
       0      .1       0  1450.9    .045       0  1485.9      .1       0
Bank Sta=1450.9,1485.9
XS Rating Curve= 0 ,0
Exp/Cntr=0.3,0.1

Type RM Length L Ch R = 1 ,37708.4 ,358.1,369,380
XS GIS Cut Line= 4
     1841189.807        346365.9     1841632.458      347059.821
     1841878.072      347333.129     1841900.938      347550.355
#Sta/Elev= 30
       0 1079.52    19.8 1069.39    29.8 1065.86    39.7  1064.3    99.2 1039.32
   148.8 1030.64   178.5 1027.88   426.4 1021.24   862.8 1019.41   991.9 1016.21
  1051.4 1010.72  1061.4  1010.7  1086.4 1010.97    1131 1017.38  1160.8 1015.73
  1170.7 1016.48  1180.6 1019.07  1190.5  1023.5  1200.5 1032.94  1210.4    1046
  1220.3 1061.02  1230.2 1071.46  1240.2 1076.09  1250.1 1089.99    1260 1101.98
  1299.8 1141.79  1319.6 1158.22  1329.5 1164.38  1339.5  1165.8    1409 1220.16
#Mann= 3 , 0 , 0
       0      .1       0  1051.4    .045       0  1086.4      .1       0
Bank Sta=1051.4,1086.4
XS Rating Curve= 0 ,0
Exp/Cntr=0.3,0.1

Type RM Length L Ch R = 1 ,37339.4 ,224.5,225.6,227.6
XS GIS Cut Line= 3
     1841027.459      346331.601     1841555.662      347598.374
     1841590.517       347938.44
#Sta/Elev= 30
       0 1175.64    19.9 1158.61    39.8 1135.67    59.7 1118.54    79.6 1109.26
   139.2 1069.18   159.1 1058.36   169.1  1057.5   208.9 1038.91   258.6 1024.95
     358 1017.41   765.8  1019.2  1054.2 1015.53  1127.1 1009.23  1153.7 1009.19
  1162.1 1010.12  1183.5 1018.24  1223.3 1026.76  1233.2 1038.61  1253.1 1068.38
    1273 1091.89    1283 1099.82  1302.9 1110.45  1421.3  1142.7  1489.7  1153.2
  1538.5 1158.04  1567.8  1163.7  1616.7 1190.96  1626.4  1191.6  1714.3 1238.51
#Mann= 3 , 0 , 0
       0     .06       0  1127.1    .045       0  1162.1     .06       0
Bank Sta=1127.1,1162.1
XS Rating Curve= 0 ,0
Exp/Cntr=0.3,0.1

Type RM Length L Ch R = 1 ,37113.8 ,354.8,363.4,371.1
XS GIS Cut Line= 3
      1840899.41      346525.961     1841252.253      347453.391
     1841431.044      347969.288
#Sta/Elev= 30
       0 1098.79    39.7 1073.27    59.5 1066.19   109.2 1034.73   148.8 1017.17
   158.8 1015.64   238.2  1013.5   396.9 1016.37   793.8 1014.53   912.9 1012.83
   972.4  1009.2   974.8  1009.2  1009.8 1009.27  1071.7 1020.52  1081.6 1027.99
  1091.6 1030.66  1121.3 1059.57  1141.2 1070.22    1161 1086.41  1190.8 1104.21
  1200.8 1106.77  1220.6  1117.2  1290.1 1146.23    1310  1151.5  1389.4 1190.48
  1409.2 1195.65  1488.6 1237.48  1498.6 1241.59  1508.5 1242.78  1538.3 1257.95
#Mann= 3 , 0 , 0
       0     .06       0   974.8    .045       0  1009.8     .06       0
Bank Sta=974.8,1009.8
XS Rating Curve= 0 ,0
Exp/Cntr=0.3,0.1

Type RM Length L Ch R = 1 ,36750.4 ,237.4,236.5,236
XS GIS Cut Line= 3
     1840700.476      346736.328     1840890.264      347461.178
     1840947.097      348037.286
#Sta/Elev= 30
       0 1053.02      10 1047.42      20 1045.25      50 1032.14    99.9 1014.01
   109.9 1012.05   289.7 1014.42   449.6 1012.18   719.3 1013.93   729.3 1013.32
   769.2 1006.64   786.3 1006.19   821.3  1006.1     919 1005.13   938.9 1005.72
   988.8 1015.94   998.8    1022  1008.8 1031.76  1018.8 1032.27  1068.7 1079.13
  1088.6 1090.16  1108.6  1098.5  1118.6 1099.04  1128.6 1102.87  1198.4 1132.98
  1208.4 1133.76  1258.3 1152.94  1298.2 1164.52  1308.2 1165.63  1328.2 1172.57
#Mann= 3 , 0 , 0
       0     .06       0   786.3    .045       0   821.3     .06       0
Bank Sta=786.3,821.3
XS Rating Curve= 0 ,0
Exp/Cntr=0.3,0.1

Type RM Length L Ch R = 1 ,36513.8 ,292.4,296.4,300.1
XS GIS Cut Line= 3
     1840558.708      346734.041     1840660.311      347539.671
     1840723.425      348082.025
#Sta/Elev= 30
       0 1094.45     9.9 1088.84    29.7 1083.12      99  1044.3   108.9  1040.5
   118.8 1038.71   138.6 1030.08     198 1011.58   356.5 1011.63   534.7 1008.91
   742.7 1010.33   752.6 1010.08   782.3 1006.33   794.5 1006.28   829.5  1006.2
   990.7 1004.52  1010.6 1006.85  1050.3  1016.7  1060.2 1021.83    1080 1035.71
    1090 1038.43  1099.9 1042.59  1119.8 1055.75  1139.6 1065.47  1169.4 1077.21
  1189.3 1080.64  1238.9  1097.3  1268.7 1108.62  1288.5 1112.52    1358 1145.06
#Mann= 3 , 0 , 0
       0     .06       0   794.5    .045       0   829.5     .06       0
Bank Sta=794.5,829.5
XS Rating Curve= 0 ,0
Exp/Cntr=0.3,0.1

Type RM Length L Ch R = 1 ,36217.4 ,343.8,348.1,352.5
XS GIS Cut Line= 3
     1840362.061      346809.499      1840375.78      347877.338
      1840375.78      348133.436
#Sta/Elev= 30
       0 1093.76      20 1084.43    29.9 1084.16    69.9 1066.83   119.8  1040.5
   129.8 1040.36   149.7 1030.92   209.6 1015.52   309.4 1008.02   419.2 1006.62
   608.8 1009.08   718.6  1007.3   758.5 1001.89   780.3 1001.22   788.5  1001.2
   815.3 1001.41   828.4 1002.57   888.3 1013.41   898.3 1013.86   908.2 1017.52
   948.2 1039.57   968.1 1046.34    1028 1052.47  1097.5  1063.1  1166.4 1087.74
  1186.1 1091.19  1215.7 1101.26  1264.9 1112.99  1284.6  1116.1    1324 1128.72
#Mann= 3 , 0 , 0
       0     .06       0   780.3    .045       0   815.3     .06       0
Bank Sta=780.3,815.3
XS Rating Curve= 0 ,0
Exp/Cntr=0.3,0.1

Type RM Length L Ch R = 1 ,35869.3 ,256.3,249.9,243.5
XS GIS Cut Line= 3
     1840030.505      346930.688     1840099.102       347083.89
      1839973.34      348073.985
#Sta/Elev= 30
       0 1096.07    39.5 1083.28    59.2 1073.08      79  1060.8    88.9 1056.62
    98.7 1055.01   167.9 1015.54   177.8 1010.41   187.8 1006.55   197.8 1005.14
   217.8    1005   307.6 1005.01   367.5 1006.51   577.1 1000.18   610.6 1000.04
     617 1000.03   636.9 1000.78   645.6 1002.71   666.9 1007.45   916.4 1011.92
   926.4 1014.96   956.3 1030.85   966.3 1032.77   976.3 1036.04   986.3 1041.02
   996.2 1043.92  1006.2 1044.65  1046.1 1043.53    1096 1040.54  1165.9 1040.48
#Mann= 3 , 0 , 0
       0     .06       0   610.6    .045       0   645.6     .06       0
Bank Sta=610.6,645.6
XS Rating Curve= 0 ,0
Exp/Cntr=0.3,0.1

Type RM Length L Ch R = 1 ,35619.4 ,386.4,366.2,346.1
XS GIS Cut Line= 3
      1839765.26      346960.414     1839785.839      347106.756
      1839845.29      348089.991
#Sta/Elev= 30
       0 1195.84    39.4 1166.81    49.3 1166.17   137.9 1103.51   147.8 1101.56
   157.7 1096.34   217.4  1055.9   227.4 1050.65   247.3 1045.91   277.1  1033.5
   326.9 1015.97   416.4 1000.86   476.1   997.7     479   997.7     496  997.83
     514  999.89   575.6 1005.88   764.7 1003.59   854.2 1006.47   884.1 1010.05
     894 1013.05   913.9 1023.19   923.9 1023.59   943.8 1026.93  1043.3 1028.47
  1083.1 1027.75    1093 1029.36    1103  1033.3  1112.9  1033.2  1132.8 1044.07
#Mann= 3 , 0 , 0
       0     .06       0     479    .045       0     514     .06       0
Bank Sta=479,514
XS Rating Curve= 0 ,0
Exp/Cntr=0.3,0.1

Type RM Length L Ch R = 1 ,35253.1 ,175.8,175.1,174.4
XS GIS Cut Line= 3
     1839177.605      347205.079     1839760.687      347920.783
     1839832.028      348112.428
#Sta/Elev= 30
       0 1207.99    59.6 1192.62    79.4 1184.51   178.7 1166.66   208.4 1156.01
   248.2 1147.57   307.7 1130.96   327.6  1120.5   367.3 1109.57   377.2 1103.99
   436.8 1057.24   456.6    1037   466.5 1034.01   486.4 1021.67   496.3 1018.84
   516.2 1003.29   526.1  997.75     546   995.6   546.4   995.6   581.4   997.8
   625.4 1005.34   823.9 1014.17   923.2 1020.97   962.1 1019.38  1030.3 1025.87
  1049.8  1033.2  1069.2 1044.25    1079 1044.86  1108.2 1054.76  1127.6 1056.91
#Mann= 3 , 0 , 0
       0     .06       0   546.4    .045       0   581.4     .06       0
Bank Sta=546.4,581.4
XS Rating Curve= 0 ,0
Exp/Cntr=0.3,0.1

Type RM Length L Ch R = 1 ,35078   ,255.7,256.6,257.5
XS GIS Cut Line= 2
     1839035.137      347324.048     1839698.948      348105.997
#Sta/Elev= 30
       0 1277.25    29.9 1259.73    49.8 1253.75    59.8  1247.9   109.5 1229.09
   159.3 1212.03   179.2  1207.1   209.1 1193.78   298.8 1123.88   308.7    1121
   328.6    1105   338.6 1099.22   348.5 1097.45   438.2 1031.02   458.1 1025.01
     488 1007.92   497.9 1003.69   517.8  997.39   532.3  994.86   557.7  994.45
   567.3  994.55   577.6  995.18   617.4 1003.24   627.4 1004.13   667.2 1004.84
   756.8 1011.66   906.2 1014.92   926.1 1017.42   985.9 1020.15  1025.7 1026.34
#Mann= 3 , 0 , 0
       0     .06       0   532.3    .045       0   567.3     .06       0
Bank Sta=532.3,567.3
XS Rating Curve= 0 ,0
Exp/Cntr=0.3,0.1

Type RM Length L Ch R = 1 ,34821.4 ,438.9,435.7,432.5
XS GIS Cut Line= 3
      1838894.92      347534.375      1839237.04      347959.843
     1839590.846      348376.025
#Sta/Elev= 30
       0 1241.21     9.9  1238.1    49.6 1211.42    59.6 1206.43    69.5 1204.88
    79.4  1199.3     129 1166.11     139 1161.27   148.9 1158.88   178.7 1135.19
   258.1 1080.52   277.9 1073.02   297.8  1056.7   347.4 1023.26   357.4 1017.68
   387.1  1006.5     407  1002.5   426.8  994.32   436.1   992.8   446.7   992.3
   471.1  992.43   486.4  994.42   506.2 1001.77   526.1 1003.98   625.4 1006.38
   814.1 1006.24   923.4 1010.74  1002.8 1025.38  1052.5 1032.49  1092.2 1042.55
#Mann= 3 , 0 , 0
       0     .06       0   436.1    .045       0   471.1     .06       0
Bank Sta=436.1,471.1
XS Rating Curve= 0 ,0
Exp/Cntr=0.3,0.1

Type RM Length L Ch R = 1 ,34385.7 ,150.5,148.7,146.8
XS GIS Cut Line= 3
     1838486.618      347802.094     1839346.813      348679.932
      1839456.57      348778.256
#Sta/Elev= 30
       0 1093.55      10 1091.74      30 1095.08    89.9 1084.71   139.9 1071.21
   169.9 1070.94   269.8 1057.77   329.7 1055.84   409.7 1044.92   449.6 1034.21
   469.6  1019.4   509.6  995.79   529.2  990.34   539.6  990.22   549.6  990.51
   564.2  994.28   579.6  999.18   599.5 1001.92   809.4  1004.2  1049.2 1003.84
  1099.1 1005.93  1129.1 1009.49  1149.1 1016.06  1179.1  1032.8  1199.1 1046.86
    1219 1068.01  1238.9 1095.96  1248.7 1103.45  1346.9 1148.56  1376.4 1159.04
#Mann= 3 , 0 , 0
       0     .06       0   529.2    .045       0   564.2     .06       0
Bank Sta=529.2,564.2
XS Rating Curve= 0 ,0
Exp/Cntr=0.3,0.1

Type RM Length L Ch R = 1 ,34237   ,241,239.7,238.3
XS GIS Cut Line= 3
     1838515.627      348071.666     1838919.329      348439.284
     1839322.173      348807.839
#Sta/Elev= 30
       0 1076.89    49.6  1065.9    69.5 1058.95   148.9  1043.9   178.7 1035.66
   258.1 1019.65     268 1015.03     278 1006.61   297.8  994.52   307.8  990.44
     325  989.37   347.5  989.25     360  990.34   367.3  991.93   387.2 1000.24
   397.1  1000.9   506.3  999.92   625.4  1003.3     824 1002.32   863.7 1004.72
   883.5 1007.51   923.2 1018.58   933.2  1025.9   943.1  1030.6     963 1047.14
  1022.5 1091.53  1042.4 1109.37  1062.2 1123.23  1082.1 1131.44    1092 1139.13
#Mann= 3 , 0 , 0
       0     .06       0     325    .045       0     360     .06       0
#XS Ineff= 2 , 0
                          655.01         1003.39
Permanent Ineff=
       F       F
Bank Sta=325,360
XS Rating Curve= 0 ,0
Exp/Cntr=0.3,0.1
